--- RICHCRK.prj (project) ---

Proj Title=RICHCRK
Current Plan=p01
Default Exp/Contr=0,0
English Units
Geom File=g01
Flow File=f01
Plan File=p01
BEGIN DESCRIPTION:
END DESCRIPTION:
DSS Export Rating Curves= 0
DSS Export Rating Curve Sorted= 0
DSS Export Volume Flow Curves= 0
DXF OffsetX= 0
DXF OffsetY= 0
DXF ScaleX= 0
DXF ScaleY= 0

--- RICHCRK.p01 (plan) ---

Plan Title=Floodplain
Program Version=4.00
Geom File=g01
Flow File=f01
K Sum by GR=0
Std Step Tol=0.01
Critical Tol=0.01
Num of Std Step Trials=20
Max Error Tol=0.3
Flow Tol Ratio=0.001
Split Flow NTrial=30
Split Flow Tol=0.02
Split Flow Ratio=0.02
Log Output Level=0
Friction Slope Method=1
Unsteady Friction Slope Method=2
Unsteady Bridges Friction Slope Method=1
Global Log Level=0
CheckData=False
Run HTab=0
Run UNet=0
Run PostProcess=0
UNET Theta=0
UNET Theta Warmup=0
UNET ZTol=0
UNET ZSATol=0
UNET MxIter=0
UNET MaxInSteps=0
UNET DtIC=0
UNET DtMin=0
UNET MaxCRTS=0
UNET WFStab=0
UNET SFStab=0
UNET WFX=0
UNET SFX=0
UNET DSS MLevel=0
UNET DZMax Abort=0
UNET Convert EG Bridges=0
UNET Use Existing IB Tables=0
UNET Froude Limit=0
UNET Froude Power=0
Write IC File=0
Echo Input=False
Echo Output=False
Write Detailed=0

--- RICHCRK.f01 (steady flow) ---

Flow Title=NFF Regression Equation
Program Version=4.00
Number of Profiles=1
Profile Names=P100yr
River Rch & RM=RICHCRK,Main      ,33096.3
953.4482
River Rch & RM=RICHCRK,Main      ,30188.9
1013.337
River Rch & RM=RICHCRK,Main      ,27904.6
1173.221
River Rch & RM=RICHCRK,Main      ,26536.8
1300.843
River Rch & RM=RICHCRK,Main      ,24724.3
1357.539
River Rch & RM=RICHCRK,Main      ,24324.3
1362.415
River Rch & RM=RICHCRK,Main      ,18329.3
1735.756
River Rch & RM=RICHCRK,Main      ,16018.6
1846.716
River Rch & RM=RICHCRK,Main      ,15177.7
2015.450
River Rch & RM=RICHCRK,Main      ,13124.3
2055.566
River Rch & RM=RICHCRK,Main      ,7098.9
2463.798
River Rch & RM=RICHCRK,Main      ,3147.9
2584.903
River Rch & RM=RICHCRK,Main      ,2747.9
2921.206
River Rch & RM=RICHCRK,Main      ,291.6
2954.798
Boundary for River Rch & Prof#=RICHCRK,Main      ,1
Up Type=0
Dn Type=3
Dn Slope=0.008146

--- RICHCRK.g01 (geometry) ---

Geom Title=USGS 10m DEM
Program Version=4.10

River Reach=RICHCRK         ,Main
Reach XY= 30
     1693918.899      255494.479     1694026.612      256101.378
     1694745.856      257085.851     1695215.768      257375.257
     1695686.317      258159.505     1696551.495      259011.943
     1697641.311      259840.143     1697932.073      260517.607
     1698205.409      262247.962     1697879.954      262860.651
     1698060.633      263713.089     1698617.729      264069.816
      1698442.84        264801.8     1698809.991      265442.286
     1698893.381      266444.132     1698570.242      267473.774
     1698126.651      267638.239     1697532.493       268372.54
     1696407.877      269271.306     1696336.069      270194.394
     1696916.328      270895.106     1697378.452      272757.497
      1696786.61      275610.152     1698212.358      277426.214
     1700205.625       278911.03     1700533.397      279647.648
     1700927.186      279860.757     1700766.439      281170.086
     1699908.211      281353.082     1699919.793      281678.537

Type RM Length L Ch R = 1 ,33096.3 ,291.2,296.3,301.4
XS GIS Cut Line= 2
      1693790.38      255556.103     1694025.275       255462.98
#Sta/Elev= 28
       0 1306.62     9.7 1305.96    19.4 1305.91    29.2 1306.33    38.9 1306.67
    48.6 1306.74    58.3 1306.54      68 1306.08    77.8 1305.07    87.5 1303.97
    97.2 1302.77   106.9 1301.38   116.6 1298.09   126.3 1296.02   135.9 1295.28
   145.8 1295.39   150.9 1296.01   155.5 1296.56   165.2  1298.6   174.9 1300.83
   184.6 1303.09   194.4 1305.85   204.1  1310.6   213.8 1320.22   223.5 1325.34
   233.2 1330.48     243 1335.67   252.7  1340.9
#Mann= 3 , 0 , 0
       0     .08       0   135.9    .045       0   150.9     .08       0
Bank Sta=135.9,150.9
XS Rating Curve= 0 ,0
Exp/Cntr=0.3,0.1

Type RM Length L Ch R = 1 ,32800   ,523.8,511.7,499.6
XS GIS Cut Line= 2
     1693819.257      255816.959     1694086.552       255776.17
#Sta/Elev= 24
       0 1331.64     9.7 1324.56    19.3 1320.73      29  1318.3    38.6    1316
    67.6  1309.6    77.2 1307.68    96.6 1304.32   106.2 1301.11   115.9 1296.85
   125.5 1293.46   135.2 1290.21   144.8 1288.28   147.9 1288.26   154.5 1288.22
   162.9 1289.42   164.2 1289.61   173.8 1291.74   183.5 1294.37   193.1 1297.64
   202.8 1302.54   212.4 1311.03   231.8 1320.39   270.4 1339.62
#Mann= 3 , 0 , 0
       0     .08       0   147.9    .045       0   162.9     .08       0
Bank Sta=147.9,162.9
XS Rating Curve= 0 ,0
Exp/Cntr=0.3,0.1

Type RM Length L Ch R = 1 ,32288.2 ,316.1,320.3,325.4
XS GIS Cut Line= 2
     1694033.352      256347.404     1694262.737      256150.538
#Sta/Elev= 27
       0 1349.26      39 1327.28    48.8 1321.93    58.5 1314.62      78 1308.19
    87.8 1303.08   107.3 1292.48     117 1287.81   126.8 1283.83   136.5 1280.71
   146.3  1278.3   152.4 1277.13     156 1276.44   165.8 1275.61   167.4 1275.83
   185.3  1278.4     195 1279.15   214.5 1282.34   224.3 1283.75     234 1285.04
   243.8 1286.84   253.5 1290.42   263.3 1295.48     273 1300.77   282.8 1307.22
   292.5  1313.3   302.3 1316.02
#Mann= 3 , 0 , 0
       0     .08       0   152.4    .045       0   167.4     .08       0
Bank Sta=152.4,167.4
XS Rating Curve= 0 ,0
Exp/Cntr=0.3,0.1

Type RM Length L Ch R = 1 ,31967.8 ,474,474.2,473.5
XS GIS Cut Line= 2
      1694206.29      256567.816     1694480.472       256413.77
#Sta/Elev= 30
       0  1330.9     9.8 1326.09    19.7 1321.97    29.5 1319.23    39.3  1317.2
    49.1 1314.26      59 1309.01    68.8 1303.45    88.4  1293.6    98.3 1284.75
   108.1 1279.61   117.9  1277.2   157.2 1271.53   163.3 1270.86   167.1 1270.44
   176.9 1270.19   178.3 1270.23   186.7 1270.47   196.6 1272.11   206.4 1275.31
   216.2 1279.59     226 1282.79   235.9 1284.54   245.7 1285.66   265.4 1286.91
   275.2 1287.82     285 1290.04   294.8  1294.2   304.7 1299.58   314.5 1307.53
#Mann= 3 , 0 , 0
       0     .08       0   163.3    .045       0   178.3     .08       0
Bank Sta=163.3,178.3
XS Rating Curve= 0 ,0
Exp/Cntr=0.3,0.1

Type RM Length L Ch R = 1 ,31493.5 ,562.2,549.6,536.9
XS GIS Cut Line= 2
     1694497.483      256936.034     1694784.614      256781.464
#Sta/Elev= 29
       0 1307.87    19.2  1298.7    28.8 1293.67    38.4 1286.32      48 1282.29
    57.6 1278.37    76.7 1271.23    86.3 1268.27   115.1 1260.11   124.7 1256.98
   128.7 1255.82   134.3  1254.2   143.7 1253.59   153.4 1255.77     163 1259.21
   172.6 1262.25   182.2 1263.88   191.8  1264.1   201.4 1264.11     211 1264.48
   220.6  1265.3   230.2  1266.3   239.8 1268.52   249.4 1277.38     259 1283.44
   268.6 1289.32   278.1  1295.3   306.9 1313.94   326.1 1326.12
#Mann= 3 , 0 , 0
       0     .08       0   128.7    .045       0   143.7     .08       0
Bank Sta=128.7,143.7
XS Rating Curve= 0 ,0
Exp/Cntr=0.3,0.1

Type RM Length L Ch R = 1 ,30943.8 ,246.5,249.4,252.4
XS GIS Cut Line= 2
     1694913.839      257385.196     1695061.096       257125.74
#Sta/Elev= 30
       0 1281.84     9.6 1279.37    38.5 1267.87    48.1 1264.28    57.7  1260.9
    67.4 1257.85      77 1256.04    86.6 1254.54    96.2 1251.96   105.9 1251.36
   115.5 1251.98   125.1 1251.37   134.7 1248.78   141.3 1246.32   144.4 1245.16
     154 1242.61   156.3 1242.57   163.6 1242.45   173.2 1242.78   182.8 1246.35
   192.5 1251.15   202.1 1255.52   221.3 1263.81     231 1268.86   240.6 1274.96
   250.2 1282.05   259.8 1285.83   269.5 1289.17   288.7 1301.46   298.3 1307.32
#Mann= 3 , 0 , 0
       0     .08       0   141.3    .045       0   156.3     .08       0
Bank Sta=141.3,156.3
XS Rating Curve= 0 ,0
Exp/Cntr=0.3,0.1

Type RM Length L Ch R = 1 ,30694.3 ,494.9,505.3,515.6
XS GIS Cut Line= 2
     1695114.952      257492.676     1695278.646      257276.352
#Sta/Elev= 27
       0 1253.65     9.7 1252.28    19.4 1251.25    29.1 1249.99    38.8 1250.64
    48.4 1252.22    58.1 1253.99    67.8 1255.64    77.5 1256.88    87.2 1256.31
    96.9 1253.46   106.6 1250.87   116.3 1249.28     126 1244.28   135.6 1239.53
   145.3 1237.57   146.4 1237.69     155 1238.64   161.4 1241.11   164.7 1242.39
   174.4 1246.78   184.1  1250.7   193.8 1253.39   203.5 1255.25   213.2 1261.07
   222.8 1269.07   271.3 1303.42
#Mann= 3 , 0 , 0
       0     .08       0   146.4    .045       0   161.4     .08       0
Bank Sta=146.4,161.4
XS Rating Curve= 0 ,0
Exp/Cntr=0.3,0.1

Type RM Length L Ch R = 1 ,30188.9 ,639.8,628.1,616.3
XS GIS Cut Line= 2
     1695379.453      257833.608     1695655.595      257694.559
#Sta/Elev= 30
       0 1261.27     9.7 1259.58    19.3 1256.63      29 1250.05    38.6 1246.69
    48.3    1244      58 1242.01    67.6 1240.74      87 1239.24    96.6 1238.28
   115.9 1235.67   125.6 1232.97   135.3 1230.51   144.9 1228.24     155  1226.5
   164.2 1226.28     170 1226.69   183.6 1227.91   193.2 1229.17   202.9 1230.61
   212.6 1232.42   222.2 1236.54   231.9 1242.04   241.5 1247.17   251.2 1254.97
   260.9 1263.19   270.5 1270.14   280.2 1276.55   299.5 1287.66   309.2 1292.77
#Mann= 3 , 0 , 0
       0     .08       0     155    .045       0     170     .08       0
Bank Sta=155,170
XS Rating Curve= 0 ,0
Exp/Cntr=0.3,0.1

Type RM Length L Ch R = 1 ,29560.6 ,459.1,465.4,471.7
XS GIS Cut Line= 2
     1695726.607      258428.753     1695919.052      258141.142
#Sta/Elev= 30
       0 1335.27     9.6 1328.98    28.8 1315.47    38.4 1313.12    48.1 1304.18
    57.7 1295.94    67.3 1288.49    76.9 1280.62    96.1 1264.43   115.4 1248.33
     125 1240.88   134.6 1238.29   144.2 1231.03   153.8 1222.72   156.2    1221
   163.4 1215.85   171.2 1213.58     173 1213.06   182.6 1213.41   192.2 1215.63
   201.9 1218.14   211.5 1219.29   221.1  1220.1   240.3 1223.37   249.9 1224.73
     298 1230.54   317.2 1231.85   326.8 1232.99   336.4 1234.53   346.1 1235.96
#Mann= 3 , 0 , 0
       0     .08       0   156.2    .045       0   171.2     .08       0
Bank Sta=156.2,171.2
XS Rating Curve= 0 ,0
Exp/Cntr=0.3,0.1

Type RM Length L Ch R = 1 ,29094.9 ,397.4,399.7,402
XS GIS Cut Line= 2
      1696061.32      258639.434     1696282.082      258457.997
#Sta/Elev= 25
       0 1237.06      19 1226.54    28.6  1223.7    38.1  1221.2    57.2 1215.81
    66.7 1213.72    76.2 1211.94    85.7 1210.95    95.2 1209.53   104.8 1207.55
   114.3 1205.49   123.8  1202.4   133.4 1199.17   137.5 1199.01   142.9  1198.8
   152.5 1199.76   161.9 1201.91   171.4 1204.31     181 1206.41     200 1212.37
   209.6 1214.61   228.6 1223.99   238.1 1230.68   247.6 1236.42   285.8 1254.74
#Mann= 3 , 0 , 0
       0     .08       0   137.5    .045       0   152.5     .08       0
Bank Sta=137.5,152.5
XS Rating Curve= 0 ,0
Exp/Cntr=0.3,0.1

Type RM Length L Ch R = 1 ,28695.3 ,435.8,428.9,421.7
XS GIS Cut Line= 2
     1696324.627      258900.666     1696587.737      258726.265
#Sta/Elev= 28
       0  1258.1    19.1 1252.76    28.7 1249.51    38.3 1245.35    47.8 1240.68
    57.4 1235.27      67 1227.16    76.5 1222.33    86.1 1217.65    95.7 1213.09
   114.8 1206.77   133.9 1196.81   143.5 1193.94     153 1193.61   153.6 1193.67
   162.6 1194.55   168.6 1195.66   172.2 1196.32   181.7 1199.06   191.3 1202.84
   200.9 1207.87     220 1218.91   239.1 1226.39   258.3 1237.88   277.4 1249.67
     287 1258.36   296.5  1265.9   315.7  1277.6
#Mann= 3 , 0 , 0
       0     .08       0   153.6    .045       0   168.6     .08       0
Bank Sta=153.6,168.6
XS Rating Curve= 0 ,0
Exp/Cntr=0.3,0.1

Type RM Length L Ch R = 1 ,28266.3 ,359.5,361.6,363.7
XS GIS Cut Line= 2
     1696628.856      259185.579       1696829.6      258959.137
#Sta/Elev= 28
       0 1201.41     9.8 1198.49    19.5 1197.97    29.3 1197.75    58.6 1197.72
    68.3 1197.79    78.1 1197.66    87.8 1196.69    97.6 1194.55   107.4 1190.89
   126.9 1188.13   136.7 1186.35   144.4 1185.85   146.4 1185.72   156.2 1187.82
   159.4 1189.72     166 1193.63   175.7 1201.46   195.2 1214.83     205 1220.06
   214.8 1222.18   224.5 1230.28   234.3 1239.38     244 1246.42   253.8  1253.3
   273.3 1266.69   292.8 1279.74   302.6  1286.1
#Mann= 3 , 0 , 0
       0     .08       0   144.4    .045       0   159.4     .08       0
Bank Sta=144.4,159.4
XS Rating Curve= 0 ,0
Exp/Cntr=0.3,0.1

Type RM Length L Ch R = 1 ,27904.6 ,411.2,409.6,408
XS GIS Cut Line= 2
     1696883.741      259420.136     1697111.994       259205.22
#Sta/Elev= 30
       0  1218.4     9.8 1214.65    19.6 1211.32    29.4 1208.29    39.2 1205.59
      49 1203.52    58.8 1201.16    78.4 1196.31    88.2 1193.77      98 1193.54
   107.8 1192.09   127.4 1186.56   137.2 1184.29     147  1182.4     153 1181.51
   156.8 1180.95   166.6 1180.83     168 1181.27   176.4 1183.94   186.2 1189.09
   195.9 1191.67   205.7 1193.76   215.5 1197.76   235.1 1206.36   254.7 1215.26
   274.3 1224.64   284.1 1230.06   293.9 1237.66   303.7 1244.04   313.5  1246.3
#Mann= 3 , 0 , 0
       0     .08       0     153    .045       0     168     .08       0
Bank Sta=153,168
XS Rating Curve= 0 ,0
Exp/Cntr=0.3,0.1

Type RM Length L Ch R = 1 ,27494.9 ,374.3,376.7,379.1
XS GIS Cut Line= 2
     1697201.578      259680.185     1697405.212      259462.767
#Sta/Elev= 30
       0 1222.48    19.2 1213.38    28.8 1208.96    38.4 1204.39      48 1198.42
    57.7 1193.63    67.3  1189.4    76.9  1185.6    86.5 1183.97   105.7 1176.98
   115.3 1174.21   118.4 1173.69   124.9 1172.59   133.4 1172.52   134.5 1172.51
   144.1 1174.08   153.8 1177.04   163.4 1179.82     173  1182.8   182.6 1185.92
   192.2 1186.74   201.8 1188.38     221 1193.41   230.6 1196.06   240.2 1198.91
   249.8  1202.8   259.4 1208.61   278.7  1221.7   288.3 1224.28   297.9 1230.55
#Mann= 3 , 0 , 0
       0      .1       0   118.4    .045       0   133.4      .1       0
Bank Sta=118.4,133.4
XS Rating Curve= 0 ,0
Exp/Cntr=0.3,0.1

Type RM Length L Ch R = 1 ,27118.2 ,576.3,581.2,586.1
XS GIS Cut Line= 2
     1697476.636      259905.232     1697694.618      259716.975
#Sta/Elev= 30
       0 1215.73     9.6 1211.05    19.2 1206.11    28.8 1201.03    38.4 1196.26
      48 1192.74    57.6 1188.74    67.2  1184.1    76.8 1180.07    86.4 1176.71
      96 1173.93   105.6 1172.29   115.2 1171.17   124.8  1170.3     144 1168.72
   149.1 1168.19   153.6 1167.73   164.1 1167.12   172.8 1166.86   182.4 1167.16
     192 1169.65   201.6 1174.16   211.2 1179.67   220.8 1184.22   230.4  1187.9
   249.6 1195.52   259.2 1199.87   268.8 1203.03   278.4 1205.45     288 1210.75
#Mann= 3 , 0 , 0
       0      .1       0   149.1    .045       0   164.1      .1       0
Bank Sta=149.1,164.1
XS Rating Curve= 0 ,0
Exp/Cntr=0.3,0.1

Type RM Length L Ch R = 1 ,26536.8 ,306.7,316.2,325.7
XS GIS Cut Line= 2
     1697691.467      260372.793     1697943.194      260232.827
#Sta/Elev= 27
       0 1209.32     9.6 1202.23    19.2 1197.31    28.8 1193.78    38.4 1190.58
    67.2 1177.09    76.8 1172.48    86.4 1167.27      96 1161.42   105.1 1157.42
   105.6  1157.2   115.2 1156.57   120.1  1157.9   124.8 1159.18   134.4 1162.08
     144 1164.05   163.2 1166.35   172.8 1167.34   182.4 1168.46     192 1170.25
   201.6 1172.44   211.2 1176.26   220.8 1184.67   230.4 1190.72     240 1196.08
   259.2  1206.6     288 1222.21
#Mann= 3 , 0 , 0
       0      .1       0   105.1    .045       0   120.1      .1       0
Bank Sta=105.1,120.1
XS Rating Curve= 0 ,0
Exp/Cntr=0.3,0.1

Type RM Length L Ch R = 1 ,26220.5 ,214.2,212.8,211.4
XS GIS Cut Line= 2
     1697778.952      260599.104      1698055.77      260574.179
#Sta/Elev= 24
       0 1224.41    19.2 1216.09    38.3 1207.44    47.9 1198.53    67.1 1188.15
    76.7 1182.66    86.3 1176.85     115 1158.84   124.6 1152.26   134.2 1145.42
   139.3 1144.22   143.8 1143.17   153.4 1144.13   154.3 1144.29   172.5 1147.47
   201.3 1152.05   210.8  1153.7   220.4 1155.53     230 1158.56   239.6 1162.55
   249.2 1165.09   258.8 1167.83   268.4 1170.81   277.9  1173.9
#Mann= 3 , 0 , 0
       0      .1       0   139.3    .045       0   154.3      .1       0
Bank Sta=139.3,154.3
XS Rating Curve= 0 ,0
Exp/Cntr=0.3,0.1

Type RM Length L Ch R = 1 ,26007.6 ,436.4,436,435.6
XS GIS Cut Line= 2
     1697801.462      260816.787      1698055.77      260778.256
#Sta/Elev= 30
       0 1214.87     9.5 1209.63      19 1204.15    28.6 1198.35    38.1 1190.98
    47.6 1179.43    57.2 1173.09    66.7 1166.83    76.2 1160.64    85.7 1154.32
    95.3 1147.28   104.8  1140.6   113.2 1137.33   114.3  1136.9   123.8 1136.46
   128.2 1136.95   133.4 1137.52   142.9 1140.52   152.4 1142.63     162 1144.18
   171.5 1145.72     181  1147.3   190.5  1149.1     200 1151.42   209.6 1154.32
   219.1 1157.51   228.6 1161.89   238.2 1167.42   247.7  1170.8   257.2 1174.18
#Mann= 3 , 0 , 0
       0      .1       0   113.2    .045       0   128.2      .1       0
Bank Sta=113.2,128.2
XS Rating Curve= 0 ,0
Exp/Cntr=0.3,0.1

Type RM Length L Ch R = 1 ,25571.8 ,444.2,447.2,450.2
XS GIS Cut Line= 2
     1697914.589      261213.284     1698163.578      261172.836
#Sta/Elev= 29
       0 1189.12     9.7 1184.61    19.4 1180.17    29.1 1175.84    38.8  1171.6
    48.5 1167.43    58.2  1163.3    67.9 1156.57    77.6 1151.26    87.3 1147.31
      97 1143.85   106.7  1141.1   116.4 1138.57   126.1 1135.78   135.8 1133.34
   138.8 1133.05   145.5 1132.39   153.8 1133.61   155.2 1133.82   164.9 1140.24
   174.6 1148.97   184.3 1153.87     194 1158.65   203.7 1163.47   213.4 1168.36
   223.2 1173.26   232.8 1178.14   242.6 1182.98   252.2 1188.49
#Mann= 3 , 0 , 0
       0      .1       0   138.8    .045       0   153.8      .1       0
Bank Sta=138.8,153.8
XS Rating Curve= 0 ,0
Exp/Cntr=0.3,0.1

Type RM Length L Ch R = 1 ,25124.3 ,401.1,399.9,398.7
XS GIS Cut Line= 2
      1697991.52      261629.616     1698259.262      261622.471
#Sta/Elev= 28
       0    1188     9.6 1184.07    19.1 1180.08    28.7 1176.18    38.3 1170.11
    47.8 1164.59      67 1156.78    86.1 1148.74    95.7 1145.07   105.2 1141.85
   124.4 1136.12   133.9 1131.88   143.5 1125.84   149.2 1125.09     153 1124.59
   162.6 1125.43   164.2  1125.8   172.2 1127.63   181.8 1130.29   191.3 1133.62
   200.9 1138.63   210.4 1144.88     220  1151.5   229.6 1164.56   239.1  1170.7
   248.7 1176.47   258.3 1181.92   267.8 1187.08
#Mann= 3 , 0 , 0
       0      .1       0   149.2    .045       0   164.2      .1       0
Bank Sta=149.2,164.2
XS Rating Curve= 0 ,0
Exp/Cntr=0.3,0.1

Type RM Length L Ch R = 1 ,24724.3 ,388.8,400.6,412.3
XS GIS Cut Line= 2
     1698063.612      262032.198     1698299.646      262013.358
#Sta/Elev= 28
       0 1145.92     9.5 1144.97    18.9 1146.12    28.4 1146.41    37.9 1144.58
    47.4 1140.88    56.8 1136.44    66.3 1131.98    75.8 1127.46    85.2 1122.45
    94.7  1117.8   103.1 1115.55   104.2 1115.26   113.7 1115.32   118.1 1115.93
   123.1 1116.62   132.6 1117.96   142.1 1119.21   151.5 1120.43     161 1121.66
   170.5 1123.13     180 1125.69   189.4 1130.27   198.9 1137.38   208.4 1149.58
   217.8 1156.48   227.3 1163.72   236.8 1171.16
#Mann= 3 , 0 , 0
       0      .1       0   103.1    .045       0   118.1      .1       0
Bank Sta=103.1,118.1
XS Rating Curve= 0 ,0
Exp/Cntr=0.3,0.1

Type RM Length L Ch R = 1 ,24324.3 ,378,374.8,371.6
XS GIS Cut Line= 2
     1698006.916      262328.229     1698254.531      262458.539
#Sta/Elev= 27
       0 1136.28     9.6  1137.5    19.3 1137.81      29 1136.74    38.6 1134.05
    48.2 1130.77    67.5 1123.67    77.2 1121.03    86.8 1119.12    96.5  1116.4
   106.1 1112.52   115.8 1109.76   125.4  1109.7   134.6 1110.31   149.6 1111.62
   154.4 1112.05     164 1114.03   173.7 1118.63   202.6 1137.23   212.3 1143.37
   221.9 1150.33   231.6 1157.76   241.2 1166.17   250.9 1172.48   260.5 1178.43
   270.2 1183.67   279.8 1190.33
#Mann= 3 , 0 , 0
       0      .1       0   134.6    .045       0   149.6      .1       0
Bank Sta=134.6,149.6
XS Rating Curve= 0 ,0
Exp/Cntr=0.3,0.1

Type RM Length L Ch R = 1 ,23948.8 ,479.1,465.3,451.5
XS GIS Cut Line= 2
     1697795.201      262652.794     1698075.533      262738.453
#Sta/Elev= 30
       0 1119.63     9.8  1115.1    19.5  1113.4    29.3 1113.13    39.1 1113.25
    48.8 1113.48    58.6 1113.42    68.4 1112.38    78.2 1110.46    87.9 1107.71
    97.7 1104.56   107.5 1102.13     115 1101.56   117.2 1101.39     127 1101.83
     130  1102.2   136.8 1103.03   146.6 1104.51   156.3 1105.82   166.1 1111.49
   175.9 1117.61   185.6 1123.85   224.7 1148.59   234.5 1154.69   244.3 1160.49
     254  1165.7   263.8 1171.23   273.6 1176.97   283.4 1181.01   293.1 1185.77
#Mann= 3 , 0 , 0
       0      .1       0     115    .045       0     130      .1       0
Bank Sta=115,130
XS Rating Curve= 0 ,0
Exp/Cntr=0.3,0.1

Type RM Length L Ch R = 1 ,23483.5 ,463,466.8,470.6
XS GIS Cut Line= 2
      1697786.56       263186.91     1698126.202      263076.246
#Sta/Elev= 30
       0  1142.7    19.3 1138.05      29 1134.39    38.6 1131.29    57.9 1126.63
    67.6 1124.74    77.2 1123.31    96.5 1120.99   106.2 1119.24   115.8 1114.83
   125.5 1099.94   135.2 1097.55   144.8 1096.84   164.1 1096.98   183.4 1096.06
   212.4 1093.84     222 1092.53   231.7 1090.83   233.3 1090.82   241.4 1090.78
   248.3 1091.91     251 1092.35   270.3 1098.74   289.6 1104.11   299.3 1108.36
   308.9 1114.35   318.6 1124.55   328.2 1132.67   347.6 1144.53   357.2 1151.09
#Mann= 3 , 0 , 0
       0      .1       0   233.3    .045       0   248.3      .1       0
Bank Sta=233.3,248.3
XS Rating Curve= 0 ,0
Exp/Cntr=0.3,0.1

Type RM Length L Ch R = 1 ,23016.6 ,378.7,364.8,350.9
XS GIS Cut Line= 2
     1697836.974      263601.003     1698154.103      263553.582
#Sta/Elev= 30
       0 1095.58     9.7 1092.81    19.4 1091.72    29.2 1090.42    48.6 1088.85
      68  1087.7   106.9 1086.46   116.6 1086.62     136 1087.84   145.8 1088.03
   155.5 1086.49   165.2 1083.51   169.1 1082.66   174.9 1081.39   184.1 1082.31
   184.6 1082.36   194.3  1088.1     204 1097.88   213.8 1111.33   223.5 1123.59
   233.2 1130.99   242.9 1138.12   252.6 1144.97   262.4 1151.56   272.1 1157.91
   281.8 1163.97   291.5 1169.82   301.2 1176.87   310.9 1186.44   320.6 1191.61
#Mann= 3 , 0 , 0
       0      .1       0   169.1    .045       0   184.1      .1       0
Bank Sta=169.1,184.1
XS Rating Curve= 0 ,0
Exp/Cntr=0.3,0.1

Type RM Length L Ch R = 1 ,22651.8 ,300.2,298.1,296.1
XS GIS Cut Line= 2
     1698095.378      263976.106     1698328.322      263752.824
#Sta/Elev= 24
       0  1084.5     9.8 1083.81    29.3 1083.58    68.4 1083.37    97.8 1083.02
   127.1 1082.52   146.7 1082.43   156.4 1082.02   166.2 1078.46     176 1073.81
   185.7 1071.65   195.6 1072.71   200.7 1073.68   205.3 1074.56   215.1  1076.6
   224.9  1078.4   244.4 1083.44   254.2 1084.19   273.8 1089.92   283.6    1093
   293.3 1096.74   303.1 1100.75   312.9 1104.84   322.7 1109.17
#Mann= 3 , 0 , 0
       0      .1       0   185.7    .045       0   200.7      .1       0
Bank Sta=185.7,200.7
XS Rating Curve= 0 ,0
Exp/Cntr=0.3,0.1

Type RM Length L Ch R = 1 ,22353.6 ,468.2,485.9,503.7
XS GIS Cut Line= 3
     1698402.542      264090.337       1698647.2      263803.453
      1698648.64      263801.764
#Sta/Elev= 30
       0 1082.72     9.7  1082.2      29 1080.82    38.7 1080.28    48.3 1079.89
    96.7 1076.49   106.3 1075.62     116 1073.01   125.7 1069.01   135.4 1067.95
     145 1067.74   154.7 1068.14     160 1068.81   164.4 1069.37     174 1070.91
   193.4  1073.5     203 1075.12   212.7 1077.14   222.4 1078.84     232 1079.68
   241.7 1080.04   251.4 1082.06   280.4 1088.32   299.7 1093.61   309.4 1096.43
     319 1099.32   328.7 1102.43     348 1104.58   367.4 1111.13   379.3  1114.8
#Mann= 3 , 0 , 0
       0      .1       0     145    .045       0     160      .1       0
Bank Sta=145,160
XS Rating Curve= 0 ,0
Exp/Cntr=0.3,0.1

Type RM Length L Ch R = 1 ,21867.6 ,491.7,490.9,490
XS GIS Cut Line= 2
     1698495.988      264406.417     1698827.888      264387.032
#Sta/Elev= 29
       0 1075.43     9.8 1073.41    19.6 1072.84    29.3 1072.15    58.7 1071.11
      88 1069.96   117.3 1068.98   136.9 1064.61     139 1064.24   146.7 1062.86
     154 1062.97   156.4    1063   166.2    1067     176 1074.56   185.8 1082.74
   195.6 1089.88   205.4 1096.62   215.1 1107.83   224.9 1115.45   234.7 1121.19
   244.5 1126.69   254.2    1132     264 1137.03   273.8 1141.79   293.4 1150.83
   303.1 1155.48   312.9 1163.86   322.7 1170.48   332.5 1175.18
#Mann= 3 , 0 , 0
       0      .1       0     139    .045       0     154      .1       0
Bank Sta=139,154
XS Rating Curve= 0 ,0
Exp/Cntr=0.3,0.1

Type RM Length L Ch R = 1 ,21376.6 ,374.7,369,363.3
XS GIS Cut Line= 2
     1698335.483      264839.595     1698616.763      264810.347
#Sta/Elev= 27
       0 1106.12    29.2  1090.9      39 1082.96    48.8 1075.78    58.5 1070.85
    68.3    1066      78 1060.96    87.8 1055.37    97.5  1050.1   107.3 1047.09
   107.7 1047.07     117 1046.61   122.7 1047.08   126.8 1047.42   136.5 1049.22
   146.3 1051.16   165.8 1053.29     195  1056.3   204.8 1057.55   214.5  1059.5
   224.3 1062.96     234 1068.06   243.8  1071.7   253.5 1074.65   263.3 1077.74
     273 1081.09   282.8 1084.69
#Mann= 3 , 0 , 0
       0      .1       0   107.7    .045       0   122.7      .1       0
Bank Sta=107.7,122.7
XS Rating Curve= 0 ,0
Exp/Cntr=0.3,0.1

Type RM Length L Ch R = 1 ,21007.5 ,281.9,283.3,284.6
XS GIS Cut Line= 2
     1698514.642      265180.218     1698796.099      265075.365
#Sta/Elev= 25
       0 1085.19     9.7 1081.27    19.4 1078.62    38.8 1073.59    48.4 1070.56
    58.1 1067.63    77.5 1062.08    87.2 1058.88    96.9 1053.63   106.6 1049.99
   116.3 1045.56     126 1042.12   135.6 1041.07   137.6 1041.13   145.3 1041.35
   152.6 1041.93   164.7 1042.99   184.1  1044.5   193.8  1045.6   222.8 1049.73
   232.5 1050.98   261.6 1057.24     281 1061.12   290.7 1064.03   300.4 1068.05
#Mann= 3 , 0 , 0
       0      .1       0   137.6    .045       0   152.6      .1       0
Bank Sta=137.6,152.6
XS Rating Curve= 0 ,0
Exp/Cntr=0.3,0.1

Type RM Length L Ch R = 1 ,20724.3 ,479.9,488.6,497.3
XS GIS Cut Line= 2
     1698654.967      265420.844     1698913.492      265341.666
#Sta/Elev= 18
       0 1100.05      29 1086.93    67.6 1067.19    86.9 1051.32    96.6 1044.17
   106.2 1038.61   115.9 1036.56     117 1036.62   125.5 1037.04     132 1037.66
   154.5 1039.96   164.2 1040.82   173.8 1042.18   193.1 1043.57   202.8 1044.15
   231.8 1045.45   260.7 1047.01   270.4  1047.7
#Mann= 3 , 0 , 0
       0      .1       0     117    .045       0     132      .1       0
Bank Sta=117,132
XS Rating Curve= 0 ,0
Exp/Cntr=0.3,0.1

Type RM Length L Ch R = 1 ,20235.8 ,321.4,311.2,301
XS GIS Cut Line= 2
     1698675.462      265846.894      1698920.97      265869.336
#Sta/Elev= 29
       0 1067.32     9.5 1060.72      19 1057.38    28.4 1054.07    37.9 1050.74
    47.4 1047.37    56.9  1043.9    66.4 1039.99    75.9 1034.97    85.3 1029.92
    94.8 1027.01    96.4 1027.19   104.3 1028.06   111.4 1029.92   113.8 1030.55
   123.3  1032.6   132.8 1033.89   142.2 1034.68   151.7 1034.96   161.2 1034.54
   170.7 1033.83   180.2 1033.44   189.6 1033.54   199.1    1034   208.6 1034.74
   218.1  1035.7   227.6 1038.18     237 1042.53   246.5 1047.73
#Mann= 3 , 0 , 0
       0      .1       0    96.4    .045       0   111.4      .1       0
Bank Sta=96.4,111.4
XS Rating Curve= 0 ,0
Exp/Cntr=0.3,0.1

Type RM Length L Ch R = 1 ,19924.3 ,386.6,400,413.3
XS GIS Cut Line= 2
     1698712.648      266196.743     1698942.113       266108.95
#Sta/Elev= 28
       0 1085.25     9.8 1076.05    19.6 1070.24    29.5 1064.86    39.3 1059.42
    49.1 1053.94      59 1048.47    68.8 1043.05    78.6 1037.61    88.4 1031.59
    98.3 1024.97   107.2 1021.24   108.1 1020.86   117.9 1021.98   122.2 1023.16
   127.8  1024.7   137.6  1027.2   147.4 1028.79   157.2 1029.34   167.1 1029.16
   176.9 1028.94   186.7 1028.92   196.6  1029.2   206.4 1029.45   216.2 1029.56
     226 1029.65   235.9 1029.75   245.7 1029.92
#Mann= 3 , 0 , 0
       0      .1       0   107.2    .045       0   122.2      .1       0
Bank Sta=107.2,122.2
XS Rating Curve= 0 ,0
Exp/Cntr=0.3,0.1

Type RM Length L Ch R = 1 ,19524.3 ,339.7,345.7,351.7
XS GIS Cut Line= 2
     1698713.359      266504.053     1698970.372      266563.404
#Sta/Elev= 30
       0 1090.92     9.8 1085.62    19.5  1080.4    29.3 1075.26    39.1 1066.15
    48.8 1060.75    58.6 1055.91    68.4  1051.1    78.2 1046.32    87.9 1041.57
    97.7 1036.86   107.5 1032.26   117.2 1027.81     127 1022.97   136.8 1016.79
   146.5 1013.87     149 1013.96   156.3 1014.23     164 1015.08   166.1 1015.31
   175.8  1016.8   185.6 1018.19   195.4 1018.99   205.2 1019.63   214.9 1020.19
   224.7 1020.96   234.5 1023.61   244.2  1029.5     254 1033.34   263.8 1037.19
#Mann= 3 , 0 , 0
       0      .1       0     149    .045       0     164      .1       0
Bank Sta=149,164
XS Rating Curve= 0 ,0
Exp/Cntr=0.3,0.1

Type RM Length L Ch R = 1 ,19178.5 ,284.9,276.8,268.8
XS GIS Cut Line= 2
     1698604.989      266790.152     1698831.343       266911.53
#Sta/Elev= 29
       0 1035.54     9.5  1032.6      19  1029.9    28.5  1027.6      38 1025.49
    47.6 1023.33    57.1 1020.96    66.6 1018.38    76.1 1015.53    85.6 1012.08
    95.1 1006.75   104.6  1003.5   114.2 1003.74   118.2 1004.22   123.7 1004.87
   133.2 1007.42   142.7 1009.07   152.2 1010.74   161.7 1012.25   171.2 1013.21
   180.7 1013.63   190.2 1013.93   199.8 1014.03   209.3 1018.45   218.8 1023.84
   228.3 1029.63   237.8 1035.24   247.3 1040.41   256.8 1044.71
#Mann= 3 , 0 , 0
       0      .1       0   118.2    .045       0   133.2      .1       0
Bank Sta=118.2,133.2
XS Rating Curve= 0 ,0
Exp/Cntr=0.3,0.1

Type RM Length L Ch R = 1 ,18901.6 ,550.8,572.3,593.8
XS GIS Cut Line= 3
     1698489.262      267084.997     1698888.992      267140.383
     1698900.418      267141.966
#Sta/Elev= 30
       0 1074.57    19.2 1061.47    28.8 1053.85    38.4 1041.68    57.6 1028.95
    86.5 1010.98    96.1 1004.16   105.7   998.5   106.6  998.29   115.3  996.24
   121.6  996.38   124.9  996.45   134.5  1000.1   144.1 1002.74   163.3 1006.65
     173 1008.05   182.6 1008.62   230.6 1008.02   240.2 1008.72   249.8 1010.85
   297.9 1026.49   317.1 1031.67   326.7 1033.83   336.3 1036.32   355.5 1038.49
   365.1 1039.81   374.7 1042.14   384.3 1044.93   393.9 1048.09   415.1 1055.86
#Mann= 3 , 0 , 0
       0      .1       0   106.6    .045       0   121.6      .1       0
Bank Sta=106.6,121.6
XS Rating Curve= 0 ,0
Exp/Cntr=0.3,0.1

Type RM Length L Ch R = 1 ,18329.3 ,415.9,404.9,394
XS GIS Cut Line= 2
     1698318.373      267397.976     1698518.578      267770.028
#Sta/Elev= 30
       0 1036.17     9.8 1029.71    19.6 1023.55      59 1000.08    68.8  999.73
    78.6  994.68    88.4  989.28    98.3   985.6   108.1  983.35   127.7  978.45
   129.5  978.36   137.6  977.98   144.5  979.13   157.2  981.51     167  982.35
   176.9  983.38   206.3  987.55   216.2  988.75     226  989.29   265.3  990.39
   275.1  990.79   294.8   991.8   334.1  994.04   363.5  994.82   373.4  995.33
   383.2  996.79     393  999.46   402.8 1003.31   412.7 1008.36   422.5 1013.99
#Mann= 3 , 0 , 0
       0      .1       0   129.5    .045       0   144.5      .1       0
Bank Sta=129.5,144.5
XS Rating Curve= 0 ,0
Exp/Cntr=0.3,0.1

Type RM Length L Ch R = 1 ,17924.3 ,640.4,646,651.7
XS GIS Cut Line= 2
     1697930.613      267649.135     1698226.203      267846.195
#Sta/Elev= 30
       0 1017.01     9.6 1012.03    19.2 1008.67    28.8 1003.19    38.4 1000.49
      48  998.82    67.2   991.3    76.8     989    86.4  986.91      96  983.89
   105.6  980.37   115.2  976.43   124.8  974.64   130.9  974.37   134.4  974.21
   145.9  975.03   172.8  978.51   182.4  979.25     192  980.52   211.2  982.23
   220.8  983.32   230.4  984.18   278.4  983.86     288  984.23   297.6  986.35
   307.2  991.06   316.8  996.92   326.4 1003.05     336 1008.39   355.2 1021.11
#Mann= 3 , 0 , 0
       0      .1       0   130.9    .045       0   145.9      .1       0
Bank Sta=130.9,145.9
XS Rating Curve= 0 ,0
Exp/Cntr=0.3,0.1

Type RM Length L Ch R = 1 ,17278.3 ,297.3,299.1,300.8
XS GIS Cut Line= 2
     1697524.473      268091.685     1697747.613      268341.138
#Sta/Elev= 27
       0 1024.17     9.6 1018.71    19.1 1013.06    28.7  1009.3    38.2 1006.86
    76.5  983.19    86.1  976.99    95.6  969.25   105.2  963.65   114.8  960.86
   118.6  960.57   124.3  960.14   133.6  960.33   143.4  960.82     153  962.43
   191.2  967.18   200.8  968.08   210.4  968.53   229.5  968.77   239.1  969.08
   267.8  970.68   277.3  971.35   286.9   972.2     306  974.07   315.6  974.92
   325.1  975.94   334.7  979.36
#Mann= 3 , 0 , 0
       0      .1       0   118.6    .045       0   133.6      .1       0
Bank Sta=118.6,133.6
XS Rating Curve= 0 ,0
Exp/Cntr=0.3,0.1

Type RM Length L Ch R = 1 ,16978.8 ,653.4,654.4,655.4
XS GIS Cut Line= 2
     1697328.559      268256.665      1697538.17       268528.14
#Sta/Elev= 30
       0  990.44     9.8  986.06    29.4  976.56    39.2  972.13      49   969.3
    58.8  968.11    78.4  966.16      98  963.99   107.8  963.73   117.6  963.19
   127.4  962.32     147   961.2   156.8  961.01   166.6  961.44   176.4  961.26
   186.2  958.45     196  956.37   205.8  956.02   210.3  956.62   215.6  957.32
   225.3  961.54   235.2  968.53     245  975.74   274.4   997.6     294 1012.32
   303.8 1019.37   313.6 1024.85   323.4 1027.72   333.2 1035.22     343 1041.22
#Mann= 3 , 0 , 0
       0     .08       0   210.3    .045       0   225.3     .08       0
Bank Sta=210.3,225.3
XS Rating Curve= 0 ,0
Exp/Cntr=0.3,0.1

Type RM Length L Ch R = 1 ,16324.3 ,308.8,305.6,302.4
XS GIS Cut Line= 2
     1696819.685      268648.813     1697014.039      268924.258
#Sta/Elev= 30
       0  963.97     9.6  961.89    19.3   960.2    28.9  958.37    38.5  956.36
    48.2  954.61    67.4  953.17      77  951.86    86.7  950.76    96.3  950.03
   115.6   949.2   163.7  947.89   173.4  947.03     183  943.72   192.6  941.22
   202.3  941.62   207.1  943.12   211.9  944.63   221.5  948.32   222.1  948.41
   231.2  949.77   240.8  950.62   260.1  955.59   269.7  957.93     289  968.45
   298.6  973.84   308.2  977.71   317.8  978.06   327.5  977.68   337.1   978.6
#Mann= 3 , 0 , 0
       0     .08       0   207.1    .045       0   222.1     .08       0
Bank Sta=207.1,222.1
XS Rating Curve= 0 ,0
Exp/Cntr=0.3,0.1

Type RM Length L Ch R = 1 ,16018.6 ,451.7,439.9,428.1
XS GIS Cut Line= 2
      1696548.55      268842.069     1696787.473      269097.164
#Sta/Elev= 30
       0  972.13     9.7  967.21    19.4     964    29.1  961.94    38.8  960.08
    48.5  958.11    87.4  949.62    97.1  947.71   106.8  946.83   116.5   946.6
   145.6  941.56   155.3  940.32     165   940.2   174.8   940.2   184.5  938.74
   194.2  935.57   202.5  934.64   203.9  934.48   213.6  934.99   217.5  935.35
   223.3  935.89     233   938.6   252.4  943.57   262.1  945.29   271.8  947.96
   281.6   953.2     301  966.17   330.1  985.22   339.8  988.41   349.5  992.48
#Mann= 3 , 0 , 0
       0     .08       0   202.5    .045       0   217.5     .08       0
Bank Sta=202.5,217.5
XS Rating Curve= 0 ,0
Exp/Cntr=0.3,0.1

Type RM Length L Ch R = 1 ,15578.7 ,406.7,400.7,394.8
XS GIS Cut Line= 2
     1696102.148      269217.283     1696572.607      269359.172
#Sta/Elev= 30
       0  955.55    29.5  941.11    39.3   937.8    49.1  936.52      59  937.09
    78.6   942.4   117.9  947.28   127.8  947.51   137.6  946.83   167.1  943.51
   196.6   942.9   206.4  941.34   216.2  938.95   235.9  933.22   245.7  931.84
   265.4  930.71     285   930.2   304.7  927.95   307.7  927.94   314.5  927.93
   322.7  929.85   334.2   933.5     344  935.12   353.8  935.05   363.6  936.05
   373.5  937.82   383.3   940.9   432.4  947.74   471.7  952.42   491.4  956.82
#Mann= 3 , 0 , 0
       0     .08       0   307.7    .045       0   322.7     .08       0
Bank Sta=307.7,322.7
XS Rating Curve= 0 ,0
Exp/Cntr=0.3,0.1

Type RM Length L Ch R = 1 ,15177.7 ,456.4,453.4,450.4
XS GIS Cut Line= 3
     1696082.978      269696.013     1696093.564      269696.372
     1696510.021      269710.464
#Sta/Elev= 30
       0 1055.36    20.3 1049.24      30 1047.14    39.7 1039.92      59 1023.84
    68.7 1015.08    97.8  987.53   107.5     979   126.9  963.92   136.6  952.72
   146.3  943.55     156  936.98   165.6  931.79   175.3  929.18     185  928.66
   243.2  928.12   252.9   926.3   262.6   922.9   272.2   920.5   277.6  920.62
   281.9  920.72   301.3  926.46     311  927.86   330.4   928.5   349.8  931.61
   359.4  934.62   398.2  948.41   407.9  950.98   417.6   952.2   427.3   952.7
#Mann= 3 , 0 , 0
       0     .08       0   262.6    .045       0   277.6     .08       0
Bank Sta=262.6,277.6
XS Rating Curve= 0 ,0
Exp/Cntr=0.3,0.1

Type RM Length L Ch R = 1 ,14724.3 ,369.4,360.5,351.5
XS GIS Cut Line= 2
     1696169.667      270173.739     1696478.602      270142.779
#Sta/Elev= 28
       0  924.77     9.7  923.71    19.4  922.88    48.5     921    58.2  920.46
    67.9  920.14    87.3  919.92      97   919.6   106.7  918.58   116.4  916.67
   126.1  914.24   135.8  912.12   145.5  910.62   154.7  909.45   164.9  908.59
   169.7  908.89   174.6  909.19   184.4  911.71     194  915.81   203.8  919.89
   213.5  920.38   223.2  920.51     262  920.25   271.7  920.07   281.4  920.32
   291.1  926.29   300.8  943.69   310.5  954.18
#Mann= 3 , 0 , 0
       0     .08       0   154.7    .045       0   169.7     .08       0
Bank Sta=154.7,169.7
XS Rating Curve= 0 ,0
Exp/Cntr=0.3,0.1

Type RM Length L Ch R = 1 ,14363.8 ,402.3,398.2,394.1
XS GIS Cut Line= 2
       1696346.3       270554.84     1696646.309      270392.203
#Sta/Elev= 30
       0  913.26    29.2   913.4    48.8  913.78    58.5  913.78      78  913.12
    87.8  912.46    97.5  910.81   107.2  908.67     117  906.84   126.8  905.68
   134.6  905.12   146.2  904.02   149.6  903.99     156  903.93   165.8  906.44
   175.5  910.56   185.2  912.18     195   912.9   224.2  914.03     234  914.69
   253.5  916.79   263.3  918.39     273  926.23   282.8  933.19   292.5  938.28
   302.3  944.56     312  952.73   321.8  960.51   331.5  968.01   341.3  975.29
#Mann= 3 , 0 , 0
       0     .08       0   134.6    .045       0   149.6     .08       0
Bank Sta=134.6,149.6
XS Rating Curve= 0 ,0
Exp/Cntr=0.3,0.1

Type RM Length L Ch R = 1 ,13965.6 ,430.8,441.2,451.6
XS GIS Cut Line= 2
     1696619.562      270860.391      1696899.01      270635.933
#Sta/Elev= 30
       0  937.94     9.7  929.67    19.4  918.68    29.1  912.29    38.8  909.52
    77.5  908.07    96.9  906.88   106.6  906.68   116.2  907.22   125.9  908.41
   135.6  908.96   145.3  907.73   164.7  903.28   174.4  902.39   193.8  901.22
   197.2   900.7   212.2   898.8   213.1   898.7   222.8  899.67   232.5   902.6
   242.2  905.94   251.9  906.93   271.2  906.97   290.6  909.11   300.3  909.73
     310  910.98   319.7  914.02   339.1  922.97   348.7  927.68   358.4  934.69
#Mann= 3 , 0 , 0
       0     .08       0   197.2    .045       0   212.2     .08       0
Bank Sta=197.2,212.2
XS Rating Curve= 0 ,0
Exp/Cntr=0.3,0.1

Type RM Length L Ch R = 1 ,13524.3 ,400.5,399.9,399.4
XS GIS Cut Line= 2
     1696767.252      271159.047     1697103.915      271084.867
#Sta/Elev= 24
       0  996.74    28.7  981.32    38.3  976.28      67  960.12    76.6  956.19
    86.2  951.59    95.8  939.51   105.3  931.37   134.1  911.18   143.6  904.35
   153.2     898   162.8  893.26   172.4   890.6   178.3  889.83     182  889.34
   191.5  889.48   193.3  889.88   201.1  891.63   210.7  894.25   220.2  895.92
   229.8   896.4     249  896.65   296.9  897.53   344.7  898.06
#Mann= 3 , 0 , 0
       0     .08       0   178.3    .045       0   193.3     .08       0
Bank Sta=178.3,193.3
XS Rating Curve= 0 ,0
Exp/Cntr=0.3,0.1

Type RM Length L Ch R = 1 ,13124.3 ,401.7,400,398.2
XS GIS Cut Line= 2
     1696816.329      271559.152     1697160.891      271476.128
#Sta/Elev= 30
       0  924.66     9.6  920.93    19.2  916.59    28.7   911.7    38.3  907.33
    57.5  900.55      67  897.39    76.6  895.16    86.2  892.81    95.8  891.33
   162.8  882.89     182   880.4   191.6  879.31   200.7  878.41   210.7  877.82
   215.7  878.43   220.3  878.99   229.9  882.07   239.5  885.67     249  887.81
   258.6  888.67   268.2  889.29   277.8  890.35   287.4  891.73     297  894.58
   306.5  899.06   316.1  904.44   325.7  910.63   335.3  916.94   354.4  929.91
#Mann= 3 , 0 , 0
       0     .08       0   200.7    .045       0   215.7     .08       0
Bank Sta=200.7,215.7
XS Rating Curve= 0 ,0
Exp/Cntr=0.3,0.1

Type RM Length L Ch R = 1 ,12724.3 ,398.4,399.9,401.5
XS GIS Cut Line= 2
     1696971.128       271946.15     1697282.682      271844.894
#Sta/Elev= 30
       0  987.06    38.5  961.82    48.2  955.24    57.8   948.3    67.4  934.81
    77.1  919.67    86.7  908.76    96.4  899.87     106  891.71   115.6  884.46
   125.3  879.72   134.9  877.54   144.5  876.08   154.2  874.99   163.8  874.33
   183.1  871.27   184.3  871.27   192.7  871.26   199.3  872.79   202.3  873.48
   221.6  880.98   231.2  883.09   240.9  884.21   250.5  885.59   260.2  887.72
   269.8   891.4     289  895.02   298.7  897.52   308.3  901.22   327.6  909.39
#Mann= 3 , 0 , 0
       0     .08       0   184.3    .045       0   199.3     .08       0
Bank Sta=184.3,199.3
XS Rating Curve= 0 ,0
Exp/Cntr=0.3,0.1

Type RM Length L Ch R = 1 ,12324.3 ,400.7,399.9,399.2
XS GIS Cut Line= 2
     1697106.659      272310.673     1697370.339      272244.752
#Sta/Elev= 29
       0  907.31    19.4  900.64    29.1  897.21    48.5  889.86    58.2  886.98
      68  885.36    77.7  884.53    87.4  883.18    97.1   880.6   106.8  876.96
   116.5  873.03   126.2  869.66   135.9   867.7   145.6  866.31   151.7  865.55
   155.3   865.1     165  866.43   166.7  866.99   174.7  869.61   184.4  873.01
   194.1  875.98   203.8  878.62   213.6  880.64   223.3   882.3     233  884.18
   242.7  886.55   252.4  889.29   262.1  893.59   271.8  896.96
#Mann= 3 , 0 , 0
       0     .08       0   151.7    .045       0   166.7     .08       0
Bank Sta=151.7,166.7
XS Rating Curve= 0 ,0
Exp/Cntr=0.3,0.1

Type RM Length L Ch R = 1 ,11924.3 ,391.8,399.8,407.9
XS GIS Cut Line= 2
     1697175.136      272709.581     1697514.822      272612.527
#Sta/Elev= 30
       0  900.44    19.6  885.51    29.4  878.59    39.2  873.51    49.1  871.88
    58.9  871.57    68.7  871.01    78.5     870    88.3  868.61   127.6  863.68
   137.4  862.84   147.2   862.6     157  861.56   161.3   860.7   166.8  859.61
   176.3  858.47   176.6  858.43   186.4  858.49   196.3  858.95   215.9  860.12
   225.7  860.82   235.5  862.36   245.3  863.76   274.8  867.75   294.4  870.14
   304.2  871.11     314  871.85   333.6  872.93   343.5   873.2   353.3  873.32
#Mann= 3 , 0 , 0
       0     .08       0   161.3    .045       0   176.3     .08       0
Bank Sta=161.3,176.3
XS Rating Curve= 0 ,0
Exp/Cntr=0.3,0.1

Type RM Length L Ch R = 1 ,11524.3 ,378.9,382.4,385.7
XS GIS Cut Line= 2
     1697165.122      273038.039     1697534.071      273066.419
#Sta/Elev= 30
       0  899.32     9.7  893.74    19.5  888.78    29.2  884.33    48.7  876.11
    58.4   872.3    68.2  868.77    77.9  865.66    87.6  861.93    97.4  859.28
   107.1  858.05   116.8   857.2   136.3  855.88   146.1  855.51   165.5  855.37
   175.3   854.3     185  852.43     188  852.21   194.8  851.72     203  852.98
   204.5  853.21   214.2  855.43     224  857.43   233.7   858.9   243.4  860.02
   253.2  860.86   282.4  862.84   292.1  863.62   340.8  865.53     370  867.53
#Mann= 3 , 0 , 0
       0     .08       0     188    .045       0     203     .08       0
Bank Sta=188,203
XS Rating Curve= 0 ,0
Exp/Cntr=0.3,0.1

Type RM Length L Ch R = 1 ,11141.8 ,291.4,290.7,290.2
XS GIS Cut Line= 2
     1697042.722      273360.874     1697423.839      273452.233
#Sta/Elev= 30
       0  897.02    29.4  880.94      49  870.75    58.8  863.39    68.6  859.55
    78.4   856.6    88.2  855.04   107.8  853.64     147   851.4   156.8  850.18
   166.6  850.16   176.4  850.68   186.2  850.16   204.5  845.48   205.8  845.16
   215.6  844.79   219.5  845.22   225.4  845.88   235.2   847.6   254.7  850.66
   264.5  851.78   303.7   853.7   313.5  854.29   333.1  856.02   342.9  857.08
   352.7   858.7   362.5  861.82   372.3  864.16   382.1  869.28   391.9  876.69
#Mann= 3 , 0 , 0
       0     .08       0   204.5    .045       0   219.5     .08       0
Bank Sta=204.5,219.5
XS Rating Curve= 0 ,0
Exp/Cntr=0.3,0.1

Type RM Length L Ch R = 1 ,10851   ,515.3,517.6,520
XS GIS Cut Line= 2
     1696914.522      273633.151     1697365.068      273724.033
#Sta/Elev= 30
       0  914.05     9.8  906.43    19.6  897.81    29.3  885.89    39.1  879.47
    48.9   873.5    58.7  867.97    78.2   857.7      88  853.03    97.8  849.97
   107.6  848.71   127.1  847.82   166.2  846.86   205.4  844.79   215.1   844.2
   224.7  842.04   234.7  840.56   239.7  840.62   244.5  840.68   254.3  841.96
     264   843.8   273.8  845.32   293.4  847.32   322.7  849.09   361.8  850.42
   371.6  850.99   381.4  851.97     401  855.84   410.7  857.48   459.6  863.77
#Mann= 3 , 0 , 0
       0     .08       0   224.7    .045       0   239.7     .08       0
Bank Sta=224.7,239.7
XS Rating Curve= 0 ,0
Exp/Cntr=0.3,0.1

Type RM Length L Ch R = 1 ,10333.4 ,479.7,479.1,478.4
XS GIS Cut Line= 2
     1696787.571      274096.449     1697200.695      274222.738
#Sta/Elev= 30
       0  881.48     9.8  874.11    19.6  866.23    29.4  860.14    39.3  854.34
    49.1  849.82    58.9  847.56    98.2  844.38   117.8  845.22   137.4   840.3
   147.3   839.5   196.4  840.16   245.4  841.46   255.3  841.59   265.1   841.3
   274.9  839.98     294  835.65   304.4  834.46     309  834.69   314.2  834.95
     324  839.48   333.8   842.4   343.6   844.5   353.4  845.78   363.3  846.25
   373.1  848.95   382.9  855.63   402.5  873.07   412.4  881.46     432  900.75
#Mann= 3 , 0 , 0
       0     .08       0     294    .045       0     309     .08       0
#XS Ineff= 2 , 0
          256.01  841.47
Permanent Ineff=
       F       F
Bank Sta=294,309
XS Rating Curve= 0 ,0
Exp/Cntr=0.3,0.1

Type RM Length L Ch R = 1 ,9854.1  ,335.4,329.7,324.1
XS GIS Cut Line= 2
     1696696.627      274563.143     1697046.011      274661.942
#Sta/Elev= 29
       0  851.22    39.2  846.65    49.1  845.59    58.9  843.59    78.5  841.51
    98.1  839.28   107.9  838.02   117.8  836.59   127.6  835.31   137.4  834.46
     157  834.07   166.8  833.42   196.3  830.73   215.9  828.72   235.5  826.59
   245.3  825.93   247.5  825.99   255.1   826.2   262.5  829.17     265  830.18
   274.8  832.69   284.6  834.54   294.4   835.7     314  836.39   323.8  840.14
   333.6  850.61   343.5  866.28   353.3  880.52   363.1  893.59
#Mann= 3 , 0 , 0
       0     .08       0   247.5    .045       0   262.5     .08       0
Bank Sta=247.5,262.5
XS Rating Curve= 0 ,0
Exp/Cntr=0.3,0.1

Type RM Length L Ch R = 1 ,9524.3  ,398.6,399.9,401.2
XS GIS Cut Line= 2
     1696683.927      274945.355     1696977.558      274952.322
#Sta/Elev= 25
       0  868.21     9.8  868.56    19.6  866.57    29.4  863.07    78.3  843.35
    97.9  835.62   107.7  829.08   117.5  826.49   137.1     825   166.4  822.17
   176.2  821.48   178.5   821.5     186  821.58   193.5  822.84   195.8  823.22
   205.6  828.05   215.4  830.81   225.2   831.7     235  832.29   244.8  833.24
   254.6  836.13   264.3  843.85   274.1   856.4   283.9  870.22   293.7  882.07
#Mann= 3 , 0 , 0
       0     .08       0   178.5    .045       0   193.5     .08       0
Bank Sta=178.5,193.5
XS Rating Curve= 0 ,0
Exp/Cntr=0.3,0.1

Type RM Length L Ch R = 1 ,9124.3  ,412.7,400,387.2
XS GIS Cut Line= 2
     1696636.961      275327.266     1696908.613      275349.904
#Sta/Elev= 26
       0  853.45     9.7  850.15    19.5     847    29.2  843.31    38.9   839.3
    58.4  830.97    68.2  826.96    77.9  823.17    87.6  820.04    97.4  818.04
   107.1  816.68   116.8  816.31   136.3  815.79     148  815.33   155.8  814.89
     163   814.8   165.5  814.77   175.2   816.6   194.7  823.01   204.4  825.36
   214.2  826.82   223.9  829.75   233.6  835.11   243.4  841.89   253.1  848.78
   272.6  862.28
#Mann= 3 , 0 , 0
       0     .08       0     148    .045       0     163     .08       0
Bank Sta=148,163
XS Rating Curve= 0 ,0
Exp/Cntr=0.3,0.1

Type RM Length L Ch R = 1 ,8724.3  ,406.1,400,393.9
XS GIS Cut Line= 2
     1696710.291      275793.404     1696925.746      275680.547
#Sta/Elev= 28
       0  827.46     9.7  827.41    19.5  828.18    29.2  828.48    38.9     827
    48.6   823.8    58.4   820.4    68.1  817.34    77.8  814.03    87.6  811.26
    97.3  809.28     107  807.66   116.8   806.6   121.9  806.61   126.5  806.61
   136.2  808.38   136.9  808.59   145.9  811.31   155.7  814.12   165.4  816.44
   175.1  818.57   184.8  820.95   194.6  823.74   204.3   824.7     214   829.7
   223.8  839.96   233.5   852.4   243.2  864.65
#Mann= 3 , 0 , 0
       0     .08       0   121.9    .045       0   136.9     .08       0
Bank Sta=121.9,136.9
XS Rating Curve= 0 ,0
Exp/Cntr=0.3,0.1

Type RM Length L Ch R = 1 ,8324.3  ,403.1,400.1,397.1
XS GIS Cut Line= 2
     1696872.327      276226.527     1697132.778      275981.862
#Sta/Elev= 30
       0   818.8      58  818.89    67.6  819.56    77.3  822.61    86.9  821.76
    96.6  817.93   106.2  813.68   115.9  811.57   125.6  810.71   135.2  810.64
   154.5  811.83   164.2  811.84   183.5  810.81   193.2  809.32   202.8  807.49
   212.5  804.86   221.7  803.48   231.8  801.51   236.7  800.98   241.4  800.47
   251.1  801.95   270.4  807.19   289.7   811.3   299.4  813.53   309.1  816.18
   318.7  817.95   328.4  819.26     338  821.18   347.7  826.67   357.4  832.81
#Mann= 3 , 0 , 0
       0     .08       0   221.7    .045       0   236.7     .08       0
Bank Sta=221.7,236.7
XS Rating Curve= 0 ,0
Exp/Cntr=0.3,0.1
